--- RUMCRK.prj (project) ---

Proj Title=RUMCRK
Current Plan=p01
Default Exp/Contr=0,0
English Units
Geom File=g01
Flow File=f01
Plan File=p01
BEGIN DESCRIPTION:
END DESCRIPTION:
DSS Export Rating Curves= 0
DSS Export Rating Curve Sorted= 0
DSS Export Volume Flow Curves= 0
DXF OffsetX= 0
DXF OffsetY= 0
DXF ScaleX= 0
DXF ScaleY= 0

--- RUMCRK.p01 (plan) ---

Plan Title=Floodplain
Program Version=4.00
Geom File=g01
Flow File=f01
K Sum by GR=0
Std Step Tol=0.01
Critical Tol=0.01
Num of Std Step Trials=20
Max Error Tol=0.3
Flow Tol Ratio=0.001
Split Flow NTrial=30
Split Flow Tol=0.02
Split Flow Ratio=0.02
Log Output Level=0
Friction Slope Method=1
Unsteady Friction Slope Method=2
Unsteady Bridges Friction Slope Method=1
Global Log Level=0
CheckData=False
Run HTab=0
Run UNet=0
Run PostProcess=0
UNET Theta=0
UNET Theta Warmup=0
UNET ZTol=0
UNET ZSATol=0
UNET MxIter=0
UNET MaxInSteps=0
UNET DtIC=0
UNET DtMin=0
UNET MaxCRTS=0
UNET WFStab=0
UNET SFStab=0
UNET WFX=0
UNET SFX=0
UNET DSS MLevel=0
UNET DZMax Abort=0
UNET Convert EG Bridges=0
UNET Use Existing IB Tables=0
UNET Froude Limit=0
UNET Froude Power=0
Write IC File=0
Echo Input=False
Echo Output=False
Write Detailed=0

--- RUMCRK.f01 (steady flow) ---

Flow Title=NFF Regression Equation
Program Version=4.10
Number of Profiles= 1
Profile Names=P100yr
River Rch & RM=RUMCRK,Main            ,37974.7
1004.888
River Rch & RM=RUMCRK,Main            ,35444.7
1079.751
River Rch & RM=RUMCRK,Main            ,33131
1167.979
River Rch & RM=RUMCRK,Main            ,31899.8
1273.303
River Rch & RM=RUMCRK,Main            ,27574.7
1410.717
River Rch & RM=RUMCRK,Main            ,27274.7
1625.726
River Rch & RM=RUMCRK,Main            ,24759.1
1727.079
River Rch & RM=RUMCRK,Main            ,18869.5
1898.923
River Rch & RM=RUMCRK,Main            ,14401.9
2109.131
River Rch & RM=RUMCRK,Main            ,14168.5
2798.688
River Rch & RM=RUMCRK,Main            ,7953.8
3037.982
River Rch & RM=RUMCRK,Main            ,7619
 3807.47
River Rch & RM=RUMCRK,Main            ,774.7
3965.906
Boundary for River Rch & Prof#=RUMCRK,Main            , 1
Up Type= 0
Dn Type= 3
Dn Slope=0.010731
DSS Import GetInterval= 0
DSS Import GetPeak= 0
DSS Import FillOption= 0

--- RUMCRK.g01 (geometry) ---

Geom Title=USGS 10m DEM
Program Version=4.10

River Reach=RUMCRK          ,Main
Reach XY= 30
     1727725.501       296548.45     1726866.115      297729.817
      1726759.56      298434.005      1726095.91      299200.735
     1724531.177      299727.718     1723978.715      299530.823
     1721866.152      300071.704     1720918.742      302547.942
     1720207.605      303004.274     1718778.383      303275.294
     1717079.298      303260.237     1716034.599      302792.323
     1715118.461      301487.028     1714411.957      300968.153
     1714241.701      300363.571     1713319.771      299165.989
     1712551.883      298976.044     1711346.193      297883.858
     1709769.879      297822.474     1708735.603      298142.138
     1707624.886      297638.319     1706294.111      297706.653
     1705490.318      296908.651     1704535.959      296745.345
     1703374.281      296026.101     1700350.213      296775.458
      1700003.91      297105.546     1699053.025      296842.634
     1698289.193      297517.885     1697787.691      297578.112

Type RM Length L Ch R = 1 ,37974.7 ,400.8,399.9,398.9
XS GIS Cut Line= 2
     1727445.439      296343.734     1727992.527      296768.325
#Sta/Elev= 30
       0 1408.68    58.5    1379    97.5 1356.07   126.8 1340.13   136.6 1333.11
   214.6  1299.2   234.1 1288.74   243.8 1283.14   253.6 1273.63   263.4 1265.11
   273.1  1260.2   282.9 1257.93   312.1 1256.39   339.8  1253.9   351.1 1253.75
   354.8 1253.89   370.6 1255.07   399.9 1258.72   458.4 1261.02   477.9 1262.54
   487.7 1263.59   497.4  1265.5   507.2 1268.24   546.2  1291.2     556 1295.92
   565.7  1298.9     595 1313.51     634 1332.07   643.8 1339.46   692.5 1368.75
#Mann= 3 , 0 , 0
       0      .1       0   339.8    .045       0   354.8     .08       0
Bank Sta=339.8,354.8
XS Rating Curve= 0 ,0
Exp/Cntr=0.3,0.1

Type RM Length L Ch R = 1 ,37574.7 ,306.2,304.4,302.6
XS GIS Cut Line= 2
     1727210.953      296684.039     1727777.484      297086.008
#Sta/Elev= 30
       0 1442.91    19.6 1433.32    58.7 1410.77      88 1397.42   107.6 1381.31
   146.8 1357.54   176.1  1338.3   205.5 1317.54     225 1300.33   234.8  1296.1
   283.7 1262.52   303.3 1247.72   313.1 1244.35     317 1244.15   322.9 1243.84
     332 1244.27   401.1 1249.28   430.5 1263.78   459.8 1271.19   469.6 1276.84
   479.4 1284.41   518.5 1304.31   528.3 1308.08   547.9 1312.02   567.5 1320.23
     587 1330.96   596.8 1340.14   606.6 1346.54   675.1 1387.36   694.6 1395.42
#Mann= 3 , 0 , 0
       0      .1       0     317    .045       0     332     .08       0
Bank Sta=317,332
XS Rating Curve= 0 ,0
Exp/Cntr=0.3,0.1

Type RM Length L Ch R = 1 ,37270.2 ,445.8,446.4,447
XS GIS Cut Line= 2
     1727011.879      296946.147     1727619.073      297309.559
#Sta/Elev= 30
       0 1426.62     9.8 1422.31    98.3 1364.37   117.9 1349.95   127.8 1340.54
   137.6 1328.86   157.2 1314.74   176.9 1303.37   196.6 1295.56   235.9 1273.76
   255.5 1259.17   265.4 1253.98   304.7 1239.15   320.1 1237.31   324.3 1237.27
   335.1  1237.7   383.3 1240.17   393.1  1242.2   442.3 1265.91   471.8 1272.28
   481.6 1277.46   491.4 1285.56   520.9 1300.62   540.6 1305.03   550.4 1309.83
   589.7 1335.06   609.4 1352.36   658.5 1384.56     688 1402.83   707.6 1410.61
#Mann= 3 , 0 , 0
       0      .1       0   320.1    .045       0   335.1     .08       0
Bank Sta=320.1,335.1
XS Rating Curve= 0 ,0
Exp/Cntr=0.3,0.1

Type RM Length L Ch R = 1 ,36823.8 ,649.8,644,638.2
XS GIS Cut Line= 2
     1726791.414      297294.706     1727399.916      297702.036
#Sta/Elev= 30
       0 1416.94    19.5    1405    68.3 1373.24    87.9 1364.32   126.9 1342.63
   214.8  1286.8   224.6 1277.81   234.3 1272.66   244.1 1269.17   292.9 1243.09
   312.4 1230.58   322.2 1227.63   324.5 1227.54     332 1227.24   339.5 1227.68
   429.6 1231.34   439.4 1233.08   449.1 1237.55   458.9 1244.86   468.6 1250.82
   478.4 1258.56   546.8 1296.73   556.5 1299.82     576 1303.71   585.8 1307.32
   595.6  1316.8   663.9 1366.26     703 1390.82   712.7 1398.71   732.2  1408.1
#Mann= 3 , 0 , 0
       0     .08       0   324.5    .045       0   339.5     .08       0
Bank Sta=324.5,339.5
XS Rating Curve= 0 ,0
Exp/Cntr=0.3,0.1

Type RM Length L Ch R = 1 ,36178.9 ,376.5,377.5,378.6
XS GIS Cut Line= 2
     1726594.245      297909.807     1727269.405      298138.507
#Sta/Elev= 30
       0 1354.62    39.1 1329.48    58.6 1314.53   146.5 1275.11   156.2 1267.67
     166 1262.63   195.3 1252.34   214.8 1244.49   224.6 1241.21   253.9 1234.22
   263.6 1230.35   302.7 1222.81     332 1216.29   338.9 1215.47   351.5 1215.06
   353.9 1215.32   371.1 1217.37   400.4 1218.74   410.1 1220.74     459 1234.96
   468.7 1240.53   478.5 1244.24   556.6  1271.6   566.4 1275.66   576.1 1281.66
   615.2 1292.91   644.5 1302.26     664 1309.11   683.6 1322.14   712.8 1333.97
#Mann= 3 , 0 , 0
       0     .08       0   338.9    .045       0   353.9     .08       0
Bank Sta=338.9,353.9
XS Rating Curve= 0 ,0
Exp/Cntr=0.3,0.1

Type RM Length L Ch R = 1 ,35801.3 ,351,356.3,361.6
XS GIS Cut Line= 2
      1726474.05      298248.136      1727140.11      298510.019
#Sta/Elev= 30
       0 1398.19    19.6 1380.17      49 1360.35    58.8 1350.92    68.6 1343.18
    88.2 1330.05   107.8 1318.96   117.6 1310.05   127.4 1302.51   186.3  1269.7
   215.7 1252.19   225.5 1242.44   254.9 1224.87   274.5 1215.21   284.3 1212.22
   333.6 1205.91   343.1 1205.49   348.6 1205.64   431.4 1210.52   460.8 1214.51
   490.2 1223.56   509.8  1232.7   529.4 1243.36     549 1259.58   558.8 1265.58
   588.2 1280.03   637.3 1309.03   647.1 1318.08   656.9 1325.46   715.7 1361.04
#Mann= 3 , 0 , 0
       0     .08       0   333.6    .045       0   348.6     .08       0
Bank Sta=333.6,348.6
XS Rating Curve= 0 ,0
Exp/Cntr=0.3,0.1

Type RM Length L Ch R = 1 ,35444.7 ,476.4,479.5,482.5
XS GIS Cut Line= 2
      1726272.51      298440.818     1726858.271      298850.446
#Sta/Elev= 30
       0  1444.4    29.4 1434.17      49 1424.58    58.8 1415.16    88.1 1395.87
    97.9 1387.87   176.2 1342.99   195.8 1326.44   225.2 1307.96   244.8 1299.31
   293.8 1269.45   303.5 1261.44   313.3 1250.79   342.7 1229.38   352.5 1220.17
   362.3  1208.5   372.1 1199.49   379.5 1197.99   381.9 1197.51   394.5 1197.73
     470 1200.77     519 1204.99   528.7  1207.7   558.1 1226.27   567.9 1236.31
   597.3 1256.86   665.8 1293.36   675.6 1300.09   685.4 1308.75   714.8 1322.14
#Mann= 3 , 0 , 0
       0     .08       0   379.5    .045       0   394.5     .08       0
Bank Sta=379.5,394.5
XS Rating Curve= 0 ,0
Exp/Cntr=0.3,0.1

Type RM Length L Ch R = 1 ,34965.4 ,382.4,388.6,394.8
XS GIS Cut Line= 2
     1725990.734      298744.209     1726518.384      299237.993
#Sta/Elev= 30
       0 1410.78    29.3 1380.82    58.6 1347.42    68.4 1338.43    78.1 1333.62
    97.7 1311.49   107.4 1298.88   117.2 1289.54     127 1287.85   244.1 1285.16
   253.9 1283.96   302.7 1252.71   312.5 1246.79   322.3 1243.24     332 1236.47
   351.6 1219.64   371.1  1197.2   380.9  1189.5   386.4  1188.7   390.6 1188.09
   401.4 1189.84   419.9 1192.69   439.5 1193.61   517.6 1191.21   566.4 1198.38
   576.2 1201.74   664.1 1251.03   683.6 1266.73   703.1 1274.48   722.7  1285.4
#Mann= 3 , 0 , 0
       0     .08       0   386.4    .045       0   401.4     .08       0
Bank Sta=386.4,401.4
XS Rating Curve= 0 ,0
Exp/Cntr=0.3,0.1

Type RM Length L Ch R = 1 ,34576.6 ,464.1,464.8,465.4
XS GIS Cut Line= 2
     1725793.326      298943.286     1726196.347      299611.228
#Sta/Elev= 30
       0 1347.61     9.8 1335.73    19.5  1325.5    68.3 1278.37      78 1274.56
    87.8 1272.98   175.5 1277.83   185.3 1277.62     195 1275.03   224.3 1260.55
   263.3 1238.26   282.8 1234.14   331.6 1205.32   341.3  1198.8   360.8  1182.5
   369.9 1178.24   380.3 1177.75   384.9  1177.9   477.8 1181.63   487.6  1184.3
   526.6 1208.08   555.8 1227.05   565.6 1227.19   614.3 1260.61   653.3 1290.19
   663.1 1294.13   672.8 1296.57   750.9 1352.51   760.6 1352.85   780.1  1365.7
#Mann= 3 , 0 , 0
       0     .08       0   369.9    .045       0   384.9     .08       0
Bank Sta=369.9,384.9
XS Rating Curve= 0 ,0
Exp/Cntr=0.3,0.1

Type RM Length L Ch R = 1 ,34111.7 ,386.4,391.4,396.5
XS GIS Cut Line= 2
     1725398.038      299113.405     1725749.882      299736.641
#Sta/Elev= 30
       0 1355.87    29.4 1330.85      49  1322.3      98 1280.44   107.8 1277.28
   137.3 1275.46   147.1 1268.27   176.5 1241.85   225.5 1206.03   235.3  1204.4
   245.1 1198.79   285.7 1171.29   294.1  1169.7   300.7 1170.39   323.5 1170.56
   352.9  1167.1   382.4 1167.31     451 1172.46   460.8 1178.67   480.4 1197.76
     500  1213.4   509.8 1220.38   519.6 1221.52   558.8 1254.77     598 1283.88
   607.8 1285.55   617.6  1291.1   686.3 1339.83   705.9 1347.15   715.7 1354.19
#Mann= 3 , 0 , 0
       0     .08       0   285.7    .045       0   300.7     .08       0
Bank Sta=285.7,300.7
XS Rating Curve= 0 ,0
Exp/Cntr=0.3,0.1

Type RM Length L Ch R = 1 ,33720   ,585.5,588.5,591.5
XS GIS Cut Line= 2
     1725096.301       299212.78     1725299.115      299899.136
#Sta/Elev= 30
       0 1399.24     9.8 1401.66    68.6 1320.68    78.4 1317.04    88.2 1306.83
      98 1293.91   107.8  1285.4   117.6  1282.8   137.3 1284.25   166.7 1278.28
   205.9 1248.44   235.3 1224.51   245.1  1223.8   294.1 1182.74   303.9 1171.99
   313.7 1163.47   320.3 1161.94   323.5  1161.2   335.3 1161.53   352.9 1163.48
     451 1163.35   519.6 1174.08   529.4 1177.66   539.2 1183.16   568.6 1202.35
   588.2 1210.63   607.8 1225.49   627.5 1236.29   656.9 1245.93   715.7 1257.58
#Mann= 3 , 0 , 0
       0     .08       0   320.3    .045       0   335.3     .08       0
Bank Sta=320.3,335.3
XS Rating Curve= 0 ,0
Exp/Cntr=0.3,0.1

Type RM Length L Ch R = 1 ,33131   ,294.9,305,315.2
XS GIS Cut Line= 2
     1724581.649       299324.81     1724700.728      300030.528
#Sta/Elev= 30
       0 1289.22    19.6 1283.32    78.4 1245.66    88.2 1241.47      98 1239.83
   166.7 1198.71   176.5 1198.22   196.1 1184.92   245.1 1154.39   254.9 1154.61
   264.7 1150.13   274.5 1148.97   333.3 1149.89   350.3  1145.8   352.9 1145.22
   365.3 1146.67   382.4  1149.9   421.6 1152.84   431.4 1156.74   441.2 1163.32
   480.4 1194.04   490.2 1197.21     500 1201.84     549 1238.59   568.6 1251.38
   588.2  1257.1   647.1 1289.28   656.9 1293.22   666.7  1294.7   715.7  1322.6
#Mann= 3 , 0 , 0
       0     .08       0   350.3    .045       0   365.3     .08       0
Bank Sta=350.3,365.3
XS Rating Curve= 0 ,0
Exp/Cntr=0.3,0.1

Type RM Length L Ch R = 1 ,32826.1 ,391.7,387.2,382.7
XS GIS Cut Line= 2
     1724459.193      299306.826     1724274.338      299967.052
#Sta/Elev= 30
       0 1269.74     9.8 1262.95    29.4 1255.87    88.2 1217.45      98 1212.58
   107.7 1210.91   137.1 1191.51   176.3 1168.18   186.1 1167.16   225.3  1146.1
   235.1 1143.82   244.9 1143.56   362.4 1149.05   375.4 1145.81   390.4 1140.11
   391.8 1139.72   401.6 1148.14   411.4 1161.39   421.2  1163.1   470.1 1197.49
   489.7 1212.43   509.3 1220.39   538.7 1244.55   568.1  1265.3   577.9 1270.56
   587.7 1271.97   636.6 1303.61   656.2 1317.83     666 1320.31   685.6 1334.76
#Mann= 3 , 0 , 0
       0     .08       0   375.4    .045       0   390.4     .08       0
Bank Sta=375.4,390.4
XS Rating Curve= 0 ,0
Exp/Cntr=0.3,0.1

Type RM Length L Ch R = 1 ,32438.7 ,547,538.8,530.5
XS GIS Cut Line= 2
     1724028.238      299137.022      1723969.55      299928.185
#Sta/Elev= 30
       0    1203     9.8 1200.74    68.6 1168.36   107.7 1157.26   195.9 1156.72
   225.3  1165.3   244.9 1162.17   264.4 1147.12   274.2 1142.24   293.8 1137.82
   342.8 1135.37     382 1138.69   390.3 1134.63   405.3 1131.72   411.4 1129.04
   421.2 1131.16   470.1 1168.39   479.9 1168.48   548.5  1220.8   558.3 1220.88
   597.4 1250.01   626.8 1268.42   636.6  1268.7   646.4 1274.38   675.8 1294.11
   705.2 1318.13     715 1319.25   724.8 1326.21   783.5 1372.34   793.3 1374.06
#Mann= 3 , 0 , 0
       0     .08       0   390.3    .045       0   405.3     .08       0
Bank Sta=390.3,405.3
XS Rating Curve= 0 ,0
Exp/Cntr=0.3,0.1

Type RM Length L Ch R = 1 ,31899.8 ,283,289.9,296.8
XS GIS Cut Line= 2
     1723414.518      299429.185     1723599.168      300047.999
#Sta/Elev= 30
       0 1177.06    29.4 1159.22    39.1 1153.82    48.9 1149.48    58.7 1146.46
    68.5 1145.82    78.3 1143.92   107.6 1136.89   127.2 1133.12     137 1131.37
   166.3 1128.18   185.9 1126.98   293.5 1129.01   303.3 1126.07   313.1 1121.04
   317.7 1120.06   322.9 1118.95   332.7 1119.52   342.5 1123.68     362 1140.78
   391.4 1162.27   401.2 1168.37     411  1169.9   479.4  1216.1   489.2 1218.45
     499 1223.36   557.7 1263.98   587.1 1277.15   616.4 1295.75   645.8 1316.62
#Mann= 3 , 0 , 0
       0      .1       0   317.7    .045       0   332.7      .1       0
Bank Sta=317.7,332.7
XS Rating Curve= 0 ,0
Exp/Cntr=0.3,0.1

Type RM Length L Ch R = 1 ,31609.8 ,535.7,531.4,527
XS GIS Cut Line= 2
     1723236.788      299469.788     1723225.017      300155.304
#Sta/Elev= 30
       0 1206.13     9.8 1201.54    19.6 1200.41    78.4 1166.32    88.2 1161.48
      98 1160.69   166.5 1127.79   195.9 1123.38   293.8 1127.17   303.6 1123.54
   313.4 1115.12   318.3 1113.34   323.2 1111.55   333.3 1111.66   342.8 1113.39
   372.2 1127.48   391.8 1134.98   401.6 1136.57     431 1136.94   440.8 1139.05
   479.9 1152.92   489.7 1153.09   509.3 1163.18   538.7 1183.29   558.3 1194.58
   568.1    1195   597.5 1208.24   636.6 1223.13   646.4 1223.64   685.6 1239.48
#Mann= 3 , 0 , 0
       0      .1       0   318.3    .045       0   333.3      .1       0
Bank Sta=318.3,333.3
XS Rating Curve= 0 ,0
Exp/Cntr=0.3,0.1

Type RM Length L Ch R = 1 ,31078   ,660.5,656.5,652.6
XS GIS Cut Line= 2
     1722681.882      299611.541     1722807.536      300285.545
#Sta/Elev= 30
       0 1235.26    39.2 1194.14    58.8 1183.84    88.2 1175.32      98 1169.68
   117.5 1154.05   146.9 1125.75   156.7 1118.86   166.5 1116.89   176.3 1110.91
   205.7 1108.14   274.2  1111.3     284 1109.92   303.6 1100.46   310.5 1098.69
   323.2 1097.81   325.5 1097.99   342.8 1101.71   362.4  1109.9   391.8 1131.06
   401.6 1133.01   411.4 1138.12   470.1 1178.96   489.7 1185.96   548.5 1228.14
   568.1 1235.39   636.6 1287.96   646.4 1294.25   656.2 1295.41   685.6 1316.52
#Mann= 3 , 0 , 0
       0      .1       0   310.5    .045       0   325.5      .1       0
Bank Sta=310.5,325.5
XS Rating Curve= 0 ,0
Exp/Cntr=0.3,0.1

Type RM Length L Ch R = 1 ,30421.4 ,386.3,375.6,365
XS GIS Cut Line= 2
     1721987.108      299697.142     1722217.177      300320.888
#Sta/Elev= 30
       0 1199.93    19.6 1194.68    29.3 1194.48    48.9 1188.73    97.8 1169.05
   117.3 1166.97   146.6 1158.12   166.2 1149.47     176 1142.42   185.8 1132.02
   195.5 1131.68   205.3 1124.59   215.1 1122.72   224.9 1116.96   244.4 1100.65
   254.2 1097.42   293.3 1093.28   308.6 1088.57   322.6 1086.96   323.6 1087.13
   371.5 1097.29     440 1151.43   449.7 1157.48   459.5 1158.81     528 1206.56
   547.5 1213.28   576.8 1233.19   625.7  1262.1   635.5 1263.46   664.8 1280.92
#Mann= 3 , 0 , 0
       0      .1       0   308.6    .045       0   323.6      .1       0
Bank Sta=308.6,323.6
XS Rating Curve= 0 ,0
Exp/Cntr=0.3,0.1

Type RM Length L Ch R = 1 ,30045.7 ,290.5,288.2,285.9
XS GIS Cut Line= 2
     1721541.821       299950.66     1722030.399      300401.529
#Sta/Elev= 30
       0 1205.94     9.8 1198.13    68.4 1170.83    78.2 1167.46   107.6 1161.29
   127.1 1154.49   146.6 1145.08   195.5 1124.11   205.3 1120.37   215.1 1118.54
     264 1095.87   293.3 1084.94   311.9 1080.81   322.6 1079.07   326.9 1079.08
   342.2 1080.24   361.7 1085.63   400.8 1086.86   410.6 1089.25   420.4 1095.59
   430.2 1100.71   449.7 1109.63   469.3 1120.04   479.1 1123.77   518.2  1150.3
   557.3 1178.29   567.1 1187.27   576.8 1193.99   596.4 1201.65   664.8 1247.26
#Mann= 3 , 0 , 0
       0      .1       0   311.9    .045       0   326.9      .1       0
Bank Sta=311.9,326.9
XS Rating Curve= 0 ,0
Exp/Cntr=0.3,0.1

Type RM Length L Ch R = 1 ,29757.3 ,398.7,390.6,382.5
XS GIS Cut Line= 2
     1721355.408      300203.827     1721885.859      300604.592
#Sta/Elev= 30
       0 1224.52    19.6 1214.74    29.3 1207.36    39.1 1203.32    78.2 1192.07
    97.8 1188.82   107.6 1185.07   136.9 1169.15   156.4 1153.37   166.2 1147.54
   185.8 1136.79   205.3 1128.49   244.4 1103.63     264  1093.4   283.5 1086.62
   312.9 1082.45   332.4 1077.04   351.5 1074.64     352 1074.59   366.5 1075.99
   381.3 1079.12   400.8 1080.91   420.4 1100.51   449.7 1121.95   469.3 1133.06
   518.2 1157.31   557.3 1183.76   625.7 1221.92   645.3 1230.71   664.8 1243.43
#Mann= 3 , 0 , 0
       0      .1       0   351.5    .045       0   366.5      .1       0
Bank Sta=351.5,366.5
XS Rating Curve= 0 ,0
Exp/Cntr=0.3,0.1

Type RM Length L Ch R = 1 ,29366.6 ,345.2,345.2,345.2
XS GIS Cut Line= 2
     1721134.516      300661.056     1721808.291      300860.393
#Sta/Elev= 30
       0  1262.2     9.8 1251.11    58.6 1225.14    78.1 1213.82    87.8 1207.75
    97.6 1198.19   107.4 1190.84   117.1  1186.3   126.9 1180.55   146.4 1164.17
   175.7 1137.35   195.2 1121.76   204.9 1109.51   234.2 1095.02   273.2  1078.3
   292.8 1073.81   312.3 1067.76   320.1 1066.82   331.8 1066.53   335.1 1066.72
   468.4 1075.78     488  1078.1   497.7 1080.98   507.5 1088.15   517.2 1097.28
   556.3 1124.86     605  1162.1   614.8 1175.16   634.3 1188.79   702.6 1232.65
#Mann= 3 , 0 , 0
       0      .1       0   320.1    .045       0   335.1      .1       0
Bank Sta=320.1,335.1
XS Rating Curve= 0 ,0
Exp/Cntr=0.3,0.1

Type RM Length L Ch R = 1 ,29021.1 ,346.8,346.8,346.7
XS GIS Cut Line= 2
     1721063.426      300998.914     1721684.896      301182.775
#Sta/Elev= 30
       0 1213.33     9.8 1204.23    19.6 1197.99    39.3 1189.39    58.9 1185.14
    68.7 1181.63    78.6 1175.52    98.2 1161.33     108 1152.22   117.8 1140.69
   196.4 1083.19     216 1070.14   245.5 1067.46   294.6 1067.34   304.4 1065.52
   316.7 1060.28     324 1057.85   331.7 1058.85   353.5 1065.64   363.3 1067.49
   392.8 1069.72   412.4 1073.14   422.2 1076.87   481.2 1102.89   530.3 1126.86
   569.5 1142.63   608.8 1160.32   618.6 1164.99   628.5 1173.94   648.1  1183.8
#Mann= 3 , 0 , 0
       0      .1       0   316.7    .045       0   331.7      .1       0
Bank Sta=316.7,331.7
XS Rating Curve= 0 ,0
Exp/Cntr=0.3,0.1

Type RM Length L Ch R = 1 ,28674.2 ,303.2,302,300.8
XS GIS Cut Line= 2
     1720971.802      301332.339     1721596.627      301517.194
#Sta/Elev= 30
       0 1206.08    29.2 1191.48    38.9 1185.09    48.6 1177.19    77.8 1169.46
    87.5 1165.81   116.7 1145.62   136.2  1129.7   145.9 1117.34   155.6 1109.23
   165.3 1104.24   194.5  1091.3   243.1 1073.87   252.9 1068.38   291.8 1060.67
   316.5 1051.83   330.7 1050.73   331.5 1050.86   340.4 1052.36   350.1 1056.08
   359.8 1058.33   437.6 1058.13   447.4 1059.63   457.1 1066.29   486.3  1078.8
   544.6 1107.09   564.1 1122.68   612.7  1151.3   632.2  1164.5   651.6 1179.19
#Mann= 3 , 0 , 0
       0      .1       0   316.5    .045       0   331.5      .1       0
Bank Sta=316.5,331.5
XS Rating Curve= 0 ,0
Exp/Cntr=0.3,0.1

Type RM Length L Ch R = 1 ,28372   ,196,195.6,195.2
XS GIS Cut Line= 2
      1720847.79      301625.062     1721485.972      301780.676
#Sta/Elev= 30
       0 1252.48     9.8 1241.44    19.6 1234.54      98 1183.76   107.8 1175.07
   117.6 1168.03   137.3 1157.74   186.3 1125.59   196.1  1117.7   205.9 1107.27
   225.5 1093.81   245.1  1082.1   264.7 1072.02   294.1  1059.7   303.9 1056.47
   323.5 1053.89   362.8 1042.67   367.3  1042.7   382.3 1044.72     402 1050.42
   470.6  1052.7   490.2 1059.68     500 1065.79   509.8 1074.82   539.2 1091.92
   568.6 1111.85   598.1 1130.18   607.9 1141.09   617.7 1147.76   656.9 1171.61
#Mann= 3 , 0 , 0
       0      .1       0   367.3    .045       0   382.3      .1       0
Bank Sta=367.3,382.3
XS Rating Curve= 0 ,0
Exp/Cntr=0.3,0.1

Type RM Length L Ch R = 1 ,28176.3 ,204.8,204.8,204.8
XS GIS Cut Line= 3
     1720847.118       301828.84     1721521.902      301980.131
     1721509.151      301982.628
#Sta/Elev= 30
       0 1211.27    19.5 1198.77    29.2 1188.19      39 1180.06    48.7  1174.5
    77.9 1166.06   116.9 1142.32   126.6 1134.04   136.4 1124.13   185.1 1092.94
   214.3 1075.93     224  1065.3   243.5 1055.15   272.7 1047.64   292.2  1039.5
   297.2 1038.44   311.7 1037.44   312.2 1037.59   331.2 1043.02   350.6 1046.71
   418.8  1048.7   428.6 1051.12     448 1058.86   477.3  1073.9   516.2  1096.6
     526 1108.11   613.6 1162.84   633.1 1181.09   691.5 1217.19   704.5 1209.14
#Mann= 3 , 0 , 0
       0      .1       0   297.2    .045       0   312.2      .1       0
Bank Sta=297.2,312.2
XS Rating Curve= 0 ,0
Exp/Cntr=0.3,0.1

Type RM Length L Ch R = 1 ,27971.4 ,216,216,215.9
XS GIS Cut Line= 3
     1720784.238      302024.192     1721479.513      302180.077
     1721487.371      302178.538
#Sta/Elev= 30
       0 1233.42     9.8 1224.47    19.5 1214.16    78.1 1175.12    87.8 1169.96
    97.6 1167.27   107.4 1163.17   117.1 1149.61   165.9 1113.02     205  1085.8
   214.7 1075.04   224.5  1067.5   253.8 1052.19   263.5 1048.62   283.1 1045.29
     311 1034.06   312.3 1033.61     326 1034.23   390.4 1042.74   478.3 1046.24
     488 1048.59   497.8 1053.11   507.6 1062.78   517.3 1069.41   595.4 1107.89
   614.9 1122.19     693 1160.71   702.8  1166.3   712.5 1176.44   720.5 1180.94
#Mann= 3 , 0 , 0
       0      .1       0     311    .045       0     326      .1       0
Bank Sta=311,326
XS Rating Curve= 0 ,0
Exp/Cntr=0.3,0.1

Type RM Length L Ch R = 1 ,27755.4 ,169.7,180.5,191.3
XS GIS Cut Line= 2
     1720746.591      302235.313     1721392.894      302380.219
#Sta/Elev= 30
       0 1245.73    19.5 1234.31      39 1221.35    58.4 1206.01    68.2 1195.11
    77.9 1181.79    87.7 1174.37   116.9 1158.27   136.4  1143.9   165.6 1121.93
   175.3 1107.95   253.2 1050.45     263 1044.94   272.7 1040.82   292.2 1033.57
   304.8 1030.28   311.7 1029.55   319.8 1030.49   340.9 1036.28   360.4 1039.46
   448.1 1042.97   564.9 1050.13   574.7 1051.58   584.4 1054.76   603.9 1064.05
   613.6 1067.72   623.4 1070.19   633.1 1071.41   652.6 1072.14   662.4 1075.26
#Mann= 3 , 0 , 0
       0      .1       0   304.8    .045       0   319.8      .1       0
Bank Sta=304.8,319.8
XS Rating Curve= 0 ,0
Exp/Cntr=0.3,0.1

Type RM Length L Ch R = 1 ,27574.7 ,291.3,300,308.6
XS GIS Cut Line= 2
     1720722.393      302251.944     1721275.343      302714.921
#Sta/Elev= 30
       0    1265     9.8 1254.03    19.5 1247.72      39  1236.4    58.5 1223.61
      78 1208.88   107.2 1184.29     117 1177.05   126.7 1172.23   136.4 1165.22
   155.9 1148.97   194.9 1112.28   214.4  1095.5   263.1 1057.88   272.9 1051.08
   282.6 1042.58   292.4 1038.21   321.6 1028.67   330.4 1027.24   331.4 1027.08
   345.4 1027.96   419.1 1038.81   506.8 1042.67   604.2 1048.72     614 1050.26
   623.7 1054.66     653 1072.59   672.4 1082.79   682.2 1088.83   721.2 1105.63
#Mann= 3 , 0 , 0
       0      .1       0   330.4    .045       0   345.4      .1       0
Bank Sta=330.4,345.4
XS Rating Curve= 0 ,0
Exp/Cntr=0.3,0.1

Type RM Length L Ch R = 1 ,27274.7 ,200.3,200.3,200.3
XS GIS Cut Line= 2
     1720587.464       302346.31     1720921.215      302970.573
#Sta/Elev= 30
       0 1237.74      59 1197.78    68.8 1195.71    78.6 1191.73     118 1164.92
   147.5 1140.27   157.3 1136.97   167.1 1132.49     236 1076.42   255.6 1068.62
     295 1038.77   304.8 1034.59   314.6  1033.2   324.4 1029.74   342.9 1020.89
   353.9 1019.94   357.9 1020.19   363.8 1020.56   383.4 1026.63   393.3  1028.8
   403.1 1029.63   530.9 1032.56   540.7 1032.91   550.6 1034.75   609.6    1061
   619.4 1066.05   629.2 1067.84   639.1 1072.54   668.6 1087.35   707.9  1110.2
#Mann= 3 , 0 , 0
       0      .1       0   342.9    .045       0   357.9      .1       0
Bank Sta=342.9,357.9
XS Rating Curve= 0 ,0
Exp/Cntr=0.3,0.1

Type RM Length L Ch R = 1 ,27074.4 ,503.5,510.1,516.8
XS GIS Cut Line= 2
     1720411.088      302440.607      1720744.84      303064.869
#Sta/Elev= 30
       0 1176.97     9.8 1170.53    19.7  1167.1    39.3  1163.8      59 1156.28
    78.6 1147.97    98.3 1137.35     118 1122.92   137.6 1111.64   206.5 1046.81
   226.1 1039.06     236  1032.6   245.8 1029.99   285.1 1028.43   314.6 1025.66
   347.4 1018.12   353.9 1017.03   362.4 1017.18   393.3 1025.91   403.1 1027.04
   462.1  1026.7   471.9 1027.33   491.6 1032.12   501.4 1032.17   540.7 1047.04
   580.1 1065.22   589.9 1065.68   678.4 1111.42   688.2 1112.86   707.9 1120.89
#Mann= 3 , 0 , 0
       0      .1       0   347.4    .045       0   362.4      .1       0
Bank Sta=347.4,362.4
XS Rating Curve= 0 ,0
Exp/Cntr=0.3,0.1

Type RM Length L Ch R = 1 ,26563.9 ,417.9,415.7,413.4
XS GIS Cut Line= 2
     1720070.648      302600.619     1720224.848      303343.139
#Sta/Elev= 30
       0  1116.5     9.7 1113.43    38.9 1084.25    77.8 1052.46    87.5  1052.7
   116.7 1032.34   126.4 1027.54   145.8 1024.95   233.3 1020.22   320.8 1018.15
   379.2  1018.5   398.6 1016.34   408.4 1012.35   418.2 1011.95   427.8 1010.56
   433.2 1011.16   437.5 1011.63   447.2 1018.68     457 1028.11   486.1 1051.28
   495.8  1054.2   505.6 1059.21   563.9 1103.22   573.6  1107.9   583.4 1110.75
   651.4  1160.8   661.1 1161.69   729.2 1213.47   738.9 1215.87   758.4 1226.96
#Mann= 3 , 0 , 0
       0     .08       0   418.2    .045       0   433.2     .08       0
Bank Sta=418.2,433.2
XS Rating Curve= 0 ,0
Exp/Cntr=0.3,0.1

Type RM Length L Ch R = 1 ,26148.1 ,370.6,372.6,374.6
XS GIS Cut Line= 2
     1719632.729      302721.843     1719862.472      303453.838
#Sta/Elev= 30
       0 1111.55    19.7 1105.31    78.7 1073.32    88.5 1068.75   108.2 1062.13
     177 1023.76   216.4 1017.66   245.9 1014.81   304.9 1012.15   393.4 1010.36
   413.1 1004.76   421.7 1003.71   422.9 1003.56   432.8 1003.94   436.7 1005.87
   442.6  1008.8   472.1 1038.78   511.5  1073.8   521.3 1081.33   531.1 1082.84
   550.8 1100.25     600 1139.66   609.8 1141.85   619.7 1147.82   678.7 1195.84
   688.5 1201.19   698.4 1204.37   708.2 1212.61   727.9  1226.3   767.2 1258.04
#Mann= 3 , 0 , 0
       0     .08       0   421.7    .045       0   436.7     .08       0
Bank Sta=421.7,436.7
XS Rating Curve= 0 ,0
Exp/Cntr=0.3,0.1

Type RM Length L Ch R = 1 ,25775.3 ,364.6,366.5,368.3
XS GIS Cut Line= 2
     1719323.897      302854.876     1719473.989      303546.661
#Sta/Elev= 30
       0 1068.11     9.8 1061.91    19.7 1061.94    49.2    1043    88.5 1023.44
    98.3 1022.63   127.8 1013.16     177 1008.18   304.8 1005.11   314.6 1004.06
   333.9  998.76   344.1  998.46   348.9  999.47   353.9 1000.52   363.8  1008.6
   373.6 1018.63   422.8 1057.89   432.6 1058.97   471.9 1091.18   501.4 1112.74
   511.2 1113.69   550.6  1143.6   580.1 1167.61   589.9 1170.34   599.7 1176.43
   629.2  1200.7   648.9 1214.78   668.6 1226.19   688.2  1233.3   707.9  1242.3
#Mann= 3 , 0 , 0
       0     .08       0   333.9    .045       0   348.9     .08       0
Bank Sta=333.9,348.9
XS Rating Curve= 0 ,0
Exp/Cntr=0.3,0.1

Type RM Length L Ch R = 1 ,25408.8 ,649.4,649.4,649.5
XS GIS Cut Line= 2
     1718978.934      302820.027     1719093.017      303672.248
#Sta/Elev= 30
       0 1130.54    19.5 1113.34    39.1 1104.57    97.7 1054.95   117.2 1046.84
   156.3 1015.11   166.1 1009.02   175.9  1006.4   263.8 1001.84   381.1  999.46
   400.6  996.95   420.1   992.2   426.2   992.6   441.2  993.91   449.4  998.79
     469 1014.44   498.3 1031.42   508.1    1036   517.8 1036.88   527.6 1040.14
   566.7 1059.61   576.5 1063.14   664.4 1081.84     684 1084.46   742.6 1101.39
   762.1 1104.26   791.4 1115.32   830.5  1133.9   840.3 1134.54   859.8 1144.18
#Mann= 3 , 0 , 0
       0     .08       0   426.2    .045       0   441.2     .08       0
Bank Sta=426.2,441.2
XS Rating Curve= 0 ,0
Exp/Cntr=0.3,0.1

Type RM Length L Ch R = 1 ,24759.1 ,315.8,318.5,321.2
XS GIS Cut Line= 2
     1718349.681       302892.21     1718463.764      303744.431
#Sta/Elev= 30
       0 1183.42    19.5 1176.16    68.4 1134.82    78.2 1133.36    87.9 1126.75
   146.6 1074.75   156.3  1071.7   166.1  1065.2   195.4 1037.11   224.7 1017.08
   244.3 1010.84   273.6  992.66   324.8  982.37   332.2   981.4   339.8  982.59
   361.5  985.73   498.3  986.57   547.2  988.44   556.9  991.37   566.7  991.46
   635.1 1055.32   644.9  1056.5   703.5 1108.32   713.3  1115.4     723    1117
   732.8 1121.77   791.4 1163.99     811 1171.28   830.5 1188.79   859.8  1211.9
#Mann= 3 , 0 , 0
       0      .1       0   324.8    .045       0   339.8     .06       0
Bank Sta=324.8,339.8
XS Rating Curve= 0 ,0
Exp/Cntr=0.3,0.1

Type RM Length L Ch R = 1 ,24440.5 ,590.5,595,599.5
XS GIS Cut Line= 2
     1718073.856      302921.806     1718084.921      303796.111
#Sta/Elev= 30
       0 1165.18    19.6 1150.74    29.5 1150.26    98.2 1099.55   108.1 1098.92
   176.8 1042.92   186.7 1042.09   255.4  987.91   275.1  983.46   304.6  982.16
   324.2   975.6   332.3  975.68   347.3  976.72   373.3  980.75   481.4  980.08
     501  981.38   510.9  985.65   569.8 1027.48   579.6 1028.78   589.5 1035.27
   648.4 1081.65   658.2 1083.17   668.1 1089.68     727 1135.14   736.8  1136.7
   746.7 1142.93   815.4 1195.96   825.2  1197.7   835.1 1203.72   874.4 1233.96
#Mann= 3 , 0 , 0
       0      .1       0   332.3    .045       0   347.3     .06       0
Bank Sta=332.3,347.3
XS Rating Curve= 0 ,0
Exp/Cntr=0.3,0.1

Type RM Length L Ch R = 1 ,23845.5 ,989.1,993.8,995.3
XS GIS Cut Line= 2
     1717555.523      302902.029     1717393.603       303755.36
#Sta/Elev= 30
       0 1166.34     9.8 1163.05    19.5 1162.49    78.1 1120.55    87.8  1118.3
    97.6  1113.1   156.2 1068.19   175.7 1060.38   234.2  1012.3     244  1006.4
   253.7 1003.63     283  976.97   292.8  972.05   341.6     973   355.9   969.4
   361.1  968.04   370.8  967.94   370.9  967.95   478.2  973.58   536.8   973.9
   585.5  979.26   614.8  980.38   653.9  985.76   673.4  994.85   722.2 1023.05
   731.9    1024   751.4 1035.81   800.2 1056.22     810 1057.78   868.6 1079.14
#Mann= 3 , 0 , 0
       0      .1       0   355.9    .045       0   370.9     .06       0
Bank Sta=355.9,370.9
XS Rating Curve= 0 ,0
Exp/Cntr=0.3,0.1

Type RM Length L Ch R = 1 ,22850.3 ,644.4,649,653.7
XS GIS Cut Line= 2
     1716796.581      302576.378     1716476.096      303332.366
#Sta/Elev= 30
       0 1111.89    19.6 1092.24    29.3 1085.42    39.1 1080.83    58.6 1078.05
    78.2 1071.76   127.1 1044.09   136.8 1043.18   156.4 1035.42   205.3 1009.43
     215  1001.4   254.2  976.62   273.7  968.27     303  961.48   332.4  956.84
   469.2  955.74   486.3  951.05   498.5  949.52   501.3  950.16   508.3  951.77
   527.9  961.51   547.4  977.06   557.2  978.14   625.6 1039.46   635.4 1045.66
   645.2 1047.97   713.6 1099.26   733.1 1106.69   801.6 1156.78   821.1 1162.48
#Mann= 3 , 0 , 0
       0      .1       0   486.3    .045       0   501.3     .06       0
Bank Sta=486.3,501.3
XS Rating Curve= 0 ,0
Exp/Cntr=0.3,0.1

Type RM Length L Ch R = 1 ,22201.1 ,239,242.3,245.6
XS GIS Cut Line= 2
      1716320.63      302346.705     1715807.882      303080.181
#Sta/Elev= 30
       0 1138.56     9.8 1133.59    19.7 1130.54    39.3  1114.7      59 1091.11
    68.8 1080.83    88.5 1062.59    98.3  1055.7     118 1047.93   186.8 1001.85
   196.7  997.84   206.5  991.02   255.7  962.59   275.4  951.83   285.2  947.94
   304.9  945.78   491.7   944.1   519.5  940.49   531.1  939.93   534.5     941
   540.9  943.02   560.6  954.17   570.4  956.14   590.1  966.12   629.4  983.14
   649.1  988.18   757.2 1008.19   835.9 1039.54   845.8 1040.24   894.9 1061.16
#Mann= 3 , 0 , 0
       0      .1       0   519.5    .045       0   534.5     .06       0
Bank Sta=519.5,534.5
XS Rating Curve= 0 ,0
Exp/Cntr=0.3,0.1

Type RM Length L Ch R = 1 ,21958.7 ,498.9,499.8,500.7
XS GIS Cut Line= 2
     1716138.946      302299.795     1715594.646      302877.603
#Sta/Elev= 30
       0 1077.19    19.6 1061.49    39.2 1048.18    58.8 1038.61    68.6 1030.63
    88.2 1017.62   127.4  994.03     147  984.83   166.6   980.2     196  967.82
   235.2  956.98   254.8  945.47   264.6  943.87     392  938.95   418.5  936.52
   433.5  934.86     441  934.79   450.8  936.97   470.4  942.98   509.6  951.39
     539  959.72   548.8  963.15   568.4  973.92   597.8  983.02   617.4     987
   666.4  989.31   676.2     992   695.8  1004.1   744.8 1019.74   793.8 1038.74
#Mann= 3 , 0 , 0
       0      .1       0   418.5    .045       0   433.5     .06       0
Bank Sta=418.5,433.5
XS Rating Curve= 0 ,0
Exp/Cntr=0.3,0.1

Type RM Length L Ch R = 1 ,21458.8 ,244.7,247.3,250
XS GIS Cut Line= 2
     1715880.408      301931.715     1715275.481      302522.492
#Sta/Elev= 30
       0 1157.14     9.8 1151.25    19.7 1140.66    39.3  1124.9    78.7  1096.9
    88.5 1090.61    98.3 1086.76   108.2 1085.32   127.8 1075.02   137.6 1066.22
   157.3 1043.41   167.1 1034.48   206.5  1008.6   216.3 1005.48     236  994.16
   245.8  987.39   265.5  967.88   304.8  939.68   324.5  934.88     362  929.62
   373.6  928.73     377  929.03   403.1  931.04   648.9  936.82   658.7  940.29
   668.6  945.42   727.6  979.43   747.2  996.09   835.7 1059.92   845.6 1064.93
#Mann= 3 , 0 , 0
       0      .1       0     362    .045       0     377     .06       0
Bank Sta=362,377
XS Rating Curve= 0 ,0
Exp/Cntr=0.3,0.1

Type RM Length L Ch R = 1 ,21211.4 ,433.9,436.4,438.9
XS GIS Cut Line= 2
     1715744.596      301780.075      1715122.69      302258.896
#Sta/Elev= 30
       0 1131.88    78.5 1084.64    88.3 1079.57   107.9 1063.22   127.5 1051.65
   196.2 1014.46     206 1007.96   215.8  998.96   225.6  994.55   255.1   976.6
   284.5  954.19   304.1  934.98     314  931.58   343.4  929.67   363.3  924.88
   372.8  923.57   378.3  923.74   402.2  925.76   461.1  927.05   529.8  930.62
   559.2  932.72   578.8   936.8   618.1  956.45   647.5  968.92     677  978.57
   696.6   983.5     726  995.51   745.6  1004.4   765.3 1016.94   784.9  1026.3
#Mann= 3 , 0 , 0
       0      .1       0   363.3    .045       0   378.3     .06       0
Bank Sta=363.3,378.3
XS Rating Curve= 0 ,0
Exp/Cntr=0.3,0.1

Type RM Length L Ch R = 1 ,20774.8 ,267.2,262.2,257.2
XS GIS Cut Line= 2
     1715520.331      301455.414     1714813.154      301884.295
#Sta/Elev= 30
       0 1139.57    68.1 1108.06    77.8 1102.28    87.6 1092.33    97.3 1089.32
   136.2 1062.52   175.1  1029.6   184.9 1018.91   194.6 1006.15   204.3  996.19
   214.1  981.26   223.8  973.63     253  959.46   291.9   936.2   301.6   929.1
   311.4   925.1   346.1  917.12     360  915.38   361.1  915.45   398.9  918.95
   603.3  922.55   651.9  924.87   671.4     928   690.8  936.91   710.3  948.59
     720  958.86   778.4 1000.45   797.9 1008.95   807.6 1015.36   827.1 1031.62
#Mann= 3 , 0 , 0
       0      .1       0   346.1    .045       0   361.1     .06       0
Bank Sta=346.1,361.1
XS Rating Curve= 0 ,0
Exp/Cntr=0.3,0.1

Type RM Length L Ch R = 1 ,20512.7 ,358.4,359,359.6
XS GIS Cut Line= 2
     1715338.553      301162.902     1714726.633      301752.936
#Sta/Elev= 30
       0 1171.82    19.5 1157.98    29.3 1154.32    68.4 1130.18   117.2 1089.04
     127 1082.12   136.8  1078.3   156.3 1057.19     215 1008.12   234.5  990.29
     254  975.98   263.8  965.84   273.6  953.55   293.1  936.08   302.9  929.38
   322.4  921.82   351.8  918.02   375.5  912.69   390.5   910.8   390.8  910.78
   410.4  914.05   605.8     921   615.6  924.49   635.1  940.33   664.4  954.82
     684  961.35   703.5  971.46   752.3  993.13   820.7 1016.14     850  1028.7
#Mann= 3 , 0 , 0
       0      .1       0   375.5    .045       0   390.5     .06       0
Bank Sta=375.5,390.5
XS Rating Curve= 0 ,0
Exp/Cntr=0.3,0.1

Type RM Length L Ch R = 1 ,20153.6 ,483.6,494.4,505.2
XS GIS Cut Line= 2
     1715080.259      300927.519     1714447.157      301505.352
#Sta/Elev= 30
       0 1159.08     9.7 1156.75    48.7  1124.6    77.9  1103.3    97.4 1083.33
   107.1 1079.34   116.9 1073.53   136.4 1057.99   194.8 1008.76   214.3  985.52
     224  981.16   233.8  974.66     302  916.65   311.7  911.82   351.8     905
   360.4  904.52   366.8  905.33   389.6  909.46   516.2  910.08   545.5  911.46
   623.4  923.51   642.9  928.65   652.6   933.4   662.4  936.13   701.3  959.58
     750  997.62   769.5 1007.38     789 1024.56   798.7 1035.65   857.2 1076.17
#Mann= 3 , 0 , 0
       0      .1       0   351.8    .045       0   366.8     .06       0
Bank Sta=351.8,366.8
XS Rating Curve= 0 ,0
Exp/Cntr=0.3,0.1

Type RM Length L Ch R = 1 ,19659.2 ,802.4,789.5,776.7
XS GIS Cut Line= 2
     1714829.927      300818.058     1714071.046      301033.827
#Sta/Elev= 30
       0 1023.84     9.7 1018.11    29.2 1000.01   107.1  950.36   116.9  937.87
   136.4  926.58   175.3  907.49   185.1  905.55   214.3  906.17   370.1  904.04
   399.4  901.88     438  894.65   438.3  894.61     448  894.65     453  895.84
   457.8  896.99   467.5  901.79     487  913.02   496.8  919.84   506.5  933.28
   555.2  969.02   584.4  988.14   603.9 1006.08   672.1 1047.55   681.8 1054.25
   691.6 1064.58     711 1076.01     750 1096.92   779.2  1114.1     789 1123.35
#Mann= 3 , 0 , 0
       0     .06       0     438    .045       0     453      .1       0
Bank Sta=438,453
XS Rating Curve= 0 ,0
Exp/Cntr=0.3,0.1

Type RM Length L Ch R = 1 ,18869.5 ,634.5,639.3,644
XS GIS Cut Line= 2
     1714458.328       299848.95     1713918.665      300450.702
#Sta/Elev= 30
       0  957.18    19.5  954.26    29.2  949.98    58.4  935.08    97.4  917.08
   107.1  916.53   126.6   909.7   136.3  907.76   175.3  902.73   194.8  901.04
   301.9  894.37     409  891.06   457.7  891.12   467.4   889.2   477.2  885.58
   486.9  883.81   489.3  884.06   496.7  884.83   504.3  888.53   516.1   892.4
   555.1  913.16   564.8  916.44     594  924.48   642.7  934.43     672  941.39
   691.4   949.6   710.9  953.22   720.6  954.18   788.8  951.65   808.3  956.08
#Mann= 3 , 0 , 0
       0     .06       0   489.3    .045       0   504.3      .1       0
Bank Sta=489.3,504.3
XS Rating Curve= 0 ,0
Exp/Cntr=0.3,0.1

Type RM Length L Ch R = 1 ,18229.8 ,319,317.9,316.9
XS GIS Cut Line= 2
     1714117.495      299458.416     1713418.442      299956.098
#Sta/Elev= 30
       0   992.5     9.8  986.94    29.2   971.7      78  947.64   107.3  938.42
   136.5  924.02   175.5   909.7   204.8  899.87   224.3  895.45   253.5   884.8
   448.6  881.78   488.1  876.84   497.3  876.67   503.1   876.9   526.6  880.34
   536.3  885.14   546.1  891.82   555.8  902.15   565.6   908.7   575.3  914.84
   594.8  923.44   653.3  960.27   663.1  970.76   672.8  977.85   711.8 1002.24
   731.4 1011.16   760.6  1028.9   780.1 1046.35   828.9 1076.13   858.1 1091.86
#Mann= 3 , 0 , 0
       0     .06       0   488.1    .045       0   503.1      .1       0
Bank Sta=488.1,503.1
XS Rating Curve= 0 ,0
Exp/Cntr=0.3,0.1

Type RM Length L Ch R = 1 ,17912   ,974.8,954.5,934.2
XS GIS Cut Line= 2
     1713920.524      299180.684     1713319.596      299664.156
#Sta/Elev= 30
       0 1016.94    19.5 1010.68    29.3 1004.94      39  997.19   107.4  961.79
   126.9   955.7   136.7   951.2   156.2  938.77   234.3  901.66   253.8  895.65
   263.6   888.7   283.1  880.32   292.9  879.23   439.3   878.8   466.5  872.81
   478.4  871.88   481.5  871.97   517.4  873.61   527.2  875.58     537  880.32
     576  909.96   585.8  916.63   595.5  920.93   605.3  930.97   615.1  939.21
   693.2 1000.14   702.9 1003.73   712.7 1010.15   722.5 1020.32   771.3    1055
#Mann= 3 , 0 , 0
       0      .1       0   466.5    .045       0   481.5      .1       0
Bank Sta=466.5,481.5
XS Rating Curve= 0 ,0
Exp/Cntr=0.3,0.1

Type RM Length L Ch R = 1 ,16956.5 ,477.7,491.3,504.6
XS GIS Cut Line= 2
     1712861.285      298482.266     1712807.383      299328.765
#Sta/Elev= 30
       0 1011.85    29.2  997.31    68.2  967.72      78  966.07    87.8  960.59
   126.7  933.79   146.2  918.17     156  915.73   185.2  905.11   224.2  888.45
     234  886.66   243.7  883.38   263.2  872.16     273   868.2   302.2  865.22
     390  863.58   423.1  858.17     429  857.84   438.1  858.55   458.2   862.7
   477.7  865.06     507  871.77   575.2   877.8   633.7  881.13   721.5  890.99
     741  898.52   750.7  904.05     780  923.84   789.7  924.06   848.2  960.39
#Mann= 3 , 0 , 0
       0     .06       0   423.1    .045       0   438.1     .06       0
Bank Sta=423.1,438.1
XS Rating Curve= 0 ,0
Exp/Cntr=0.3,0.1

Type RM Length L Ch R = 1 ,16465.6 ,495.8,502,508.3
XS GIS Cut Line= 2
     1712706.026      298383.031     1712245.414      299141.047
#Sta/Elev= 30
       0  992.49    19.5  983.35    48.7  959.79    87.7  923.91    97.5  917.36
   107.2  914.63   126.7  900.15   146.2  889.28   175.4  878.54   185.2  876.35
   214.4  875.12   253.4  860.27   263.2   859.5   438.6  857.92   553.4  850.67
   555.6  850.52   568.4  851.92   575.1  854.48   623.8  894.22   633.6   896.2
   643.3  902.77   672.6  926.12     692  944.69   711.5  960.44     731   968.9
     809 1026.16   818.8  1027.7   828.5 1033.63     848 1049.28     887 1075.19
#Mann= 3 , 0 , 0
       0     .06       0   553.4    .045       0   568.4     .06       0
Bank Sta=553.4,568.4
XS Rating Curve= 0 ,0
Exp/Cntr=0.3,0.1

Type RM Length L Ch R = 1 ,15963.5 ,384.6,381.8,379
XS GIS Cut Line= 2
     1712416.303      298183.902     1711821.473      298736.508
#Sta/Elev= 30
       0 1003.32    29.4  981.18    48.9  972.28    78.3   948.3   117.4  926.63
     137  918.13   166.3  918.88   176.1  913.82   195.6  895.27   254.3  855.49
   273.9  852.02   293.5  853.18     450  850.47   479.3  844.59   482.6  844.67
   489.1  844.83   497.6  847.96   528.2  871.07   547.8  888.69   567.4  902.12
   586.9  910.58   645.6  950.39   665.2  969.11   684.7  983.51   704.3  992.53
   714.1  999.46     763  1037.1   782.6  1055.9   802.1  1063.6   811.9 1069.85
#Mann= 3 , 0 , 0
       0     .06       0   482.6    .045       0   497.6     .06       0
Bank Sta=482.6,497.6
XS Rating Curve= 0 ,0
Exp/Cntr=0.3,0.1

Type RM Length L Ch R = 1 ,15581.6 ,469,467.3,465.6
XS GIS Cut Line= 2
     1712226.821      297743.277     1711672.233      298406.459
#Sta/Elev= 30
       0 1085.21    58.9 1047.11    68.8 1041.89    78.6 1040.39   108.1 1022.81
   117.9 1016.74   137.5 1000.64     167  979.09   186.7  970.49     226  935.35
   255.4  904.36   275.1  888.96   353.7  856.93     393  844.52   402.8  843.82
   520.7  842.02   579.6   845.4   607.6  839.56   618.9  838.16   622.6  839.34
   628.7  841.29   658.2  866.41     668  868.78   677.8  874.42   746.6  918.75
   756.4  923.65   766.3  925.54   795.7  946.22   844.9  977.27   864.5   985.9
#Mann= 3 , 0 , 0
       0     .06       0   607.6    .045       0   622.6     .06       0
#XS Ineff= 2 , 0
           569.3  845.42
Permanent Ineff=
       F       F
Bank Sta=607.6,622.6
XS Rating Curve= 0 ,0
Exp/Cntr=0.3,0.1

Type RM Length L Ch R = 1 ,15114.3 ,725.7,712.1,698.6
XS GIS Cut Line= 2
     1711867.849      297361.875     1711369.171      298060.756
#Sta/Elev= 30
       0 1119.66    19.5 1106.61      39 1099.15   107.3 1055.94   117.1 1054.35
   126.8 1050.32   204.9  1005.7   214.6 1004.95   224.4  999.92   234.2  991.25
   282.9  938.29   302.4  919.65   312.2   917.3   351.2   883.8     361  877.73
     400  868.16   429.3  852.73   468.3  840.15   478.1  838.69   653.7  838.77
   692.7  831.44   697.5  832.36   702.4  833.29   712.5  840.09     761  874.92
   770.8  877.24   780.5   883.1   790.3  890.73   809.8  909.52   858.6  944.54
#Mann= 3 , 0 , 0
       0     .06       0   697.5    .045       0   712.5     .06       0
Bank Sta=697.5,712.5
XS Rating Curve= 0 ,0
Exp/Cntr=0.3,0.1

Type RM Length L Ch R = 1 ,14401.9 ,232.8,233.4,233.9
XS GIS Cut Line= 2
     1710774.021      297229.876      1710761.24      297994.306
#Sta/Elev= 30
       0 1019.88    29.4 1011.53      49 1004.94    58.8 1000.44    68.6  993.14
    78.4  989.79    88.2  984.05   117.6  958.18     147  937.73   166.6   931.5
   225.4  895.06     245  889.12   303.8  858.35   323.5  853.18   352.9  838.31
   362.7  834.46   382.3  831.71   578.3  827.73   588.1   826.6   607.7  820.36
   610.5  820.44   617.5  820.63   625.5  824.04   637.1  829.26   646.9  831.67
   705.7  868.27   715.5  872.38   725.3  874.34   754.7  892.49   764.5  899.72
#Mann= 3 , 0 , 0
       0     .06       0   610.5    .045       0   625.5     .06       0
Bank Sta=610.5,625.5
XS Rating Curve= 0 ,0
Exp/Cntr=0.3,0.1

Type RM Length L Ch R = 1 ,14168.5 ,268.3,268.3,268.3
XS GIS Cut Line= 2
      1710552.19      297315.017     1710520.713      298080.735
#Sta/Elev= 30
       0  988.11    19.6  976.09    49.1  961.04      59  956.96    68.8  955.32
   137.6  910.46   147.4  908.78     167  896.45   206.3  876.35   216.2   872.6
     226  871.46   294.8  835.77   304.6  834.75   314.4  830.36   324.2  828.48
   491.3  824.21   520.7  816.41   521.2  816.46   536.2  817.93   540.4  818.32
   599.3  856.41   609.2  861.28     619  861.72   628.8   865.5   638.6  872.27
   658.3  889.73   687.8  910.55   697.6   911.2   717.2  922.35   766.4  944.23
#Mann= 3 , 0 , 0
       0     .06       0   521.2    .045       0   536.2     .06       0
Bank Sta=521.2,536.2
XS Rating Curve= 0 ,0
Exp/Cntr=0.3,0.1

Type RM Length L Ch R = 1 ,13900.3 ,401.7,401.7,401.7
XS GIS Cut Line= 2
     1710280.604      297392.741     1710249.127       298158.46
#Sta/Elev= 30
       0  980.34    39.3  965.68    49.1  964.99    78.6  950.17    88.4  943.22
   117.9  917.21   127.7  915.81   186.7  865.14   196.5  858.18   206.3  857.17
   245.6  826.95   255.5  824.63   284.9  825.59   334.1  822.39     393  821.87
   402.8   820.3   422.5  813.85   429.7  813.86   444.7  815.07   510.9  845.75
   540.4  849.08   550.2   852.6   589.5  872.73   599.3  872.82   628.8  882.35
   668.1  905.07   677.9  905.09   746.7  943.97   756.5     944   766.4  950.17
#Mann= 3 , 0 , 0
       0     .06       0   429.7    .045       0   444.7     .06       0
Bank Sta=429.7,444.7
XS Rating Curve= 0 ,0
Exp/Cntr=0.3,0.1

Type RM Length L Ch R = 1 ,13498.5 ,5282.5,5287.3,5292.1
XS GIS Cut Line= 4
     1709878.892      297390.176     1709847.415      298155.895
     1709837.151      298405.558     1709829.822       298583.85
#Sta/Elev= 30
       0  981.55     9.8  973.46    19.6  972.76    88.4   917.5    98.2  916.66
     167  863.38   176.8  862.39   196.5  851.84     226  847.82   245.6  838.72
   255.5  838.06   294.8  821.52   334.1     821   383.2  816.85   425.5  810.14
   432.3  809.11   440.5  809.85   481.4  828.46   491.3   829.4   520.7  840.16
   550.2  837.62   589.5  839.16   628.8   855.6   668.1  861.71   727.1  877.23
   795.2  906.47   881.7  930.88   929.7     941     997  948.24  1194.7  955.69
#Mann= 3 , 0 , 0
       0     .06       0   425.5    .045       0   440.5     .06       0
Bank Sta=425.5,440.5
XS Rating Curve= 0 ,0
Exp/Cntr=0.3,0.1

Type RM Length L Ch R = 1 ,8210.5  ,255.5,256.7,257.9
XS GIS Cut Line= 4
     1705633.443      296607.625     1705152.021      296841.041
     1705054.764      297259.247     1704888.112      297975.851
#Sta/Elev= 30
       0   850.5    77.8  816.17   175.1  763.14   262.6  763.38   301.6  780.52
   505.8  782.13   544.8  777.08   603.3  747.39   621.2  746.07   622.8  746.03
   636.2  749.11   710.7  757.37     740  794.12   769.2  812.72   788.7  819.31
     857  863.05   866.8  863.75   935.1  908.28   964.4  918.58  1101.7  906.59
  1229.2   876.9  1258.7  883.09  1366.6  924.25  1425.4  949.83  1494.1  989.27
  1503.9  988.68  1572.6  1039.2  1592.2 1044.97  1651.1 1088.19  1700.1 1111.21
#Mann= 3 , 0 , 0
       0      .1       0   621.2    .045       0   636.2      .1       0
Bank Sta=621.2,636.2
XS Rating Curve= 0 ,0
Exp/Cntr=0.3,0.1
